--- RichCreek.prj (project) ---

Proj Title=RichCreek
Current Plan=p01
Default Exp/Contr=0,0
English Units
Geom File=g01
Flow File=f01
Plan File=p01
BEGIN DESCRIPTION:
END DESCRIPTION:
DSS Export Rating Curves= 0
DSS Export Rating Curve Sorted= 0
DSS Export Volume Flow Curves= 0
DXF OffsetX= 0
DXF OffsetY= 0
DXF ScaleX= 0
DXF ScaleY= 0

--- RichCreek.p01 (plan) ---

Plan Title=Floodplain
Program Version=4.00
Geom File=g01
Flow File=f01
K Sum by GR=0
Std Step Tol=0.01
Critical Tol=0.01
Num of Std Step Trials=20
Max Error Tol=0.3
Flow Tol Ratio=0.001
Split Flow NTrial=30
Split Flow Tol=0.02
Split Flow Ratio=0.02
Log Output Level=0
Friction Slope Method=1
Unsteady Friction Slope Method=2
Unsteady Bridges Friction Slope Method=1
Global Log Level=0
CheckData=False
Run HTab=0
Run UNet=0
Run PostProcess=0
UNET Theta=0
UNET Theta Warmup=0
UNET ZTol=0
UNET ZSATol=0
UNET MxIter=0
UNET MaxInSteps=0
UNET DtIC=0
UNET DtMin=0
UNET MaxCRTS=0
UNET WFStab=0
UNET SFStab=0
UNET WFX=0
UNET SFX=0
UNET DSS MLevel=0
UNET DZMax Abort=0
UNET Convert EG Bridges=0
UNET Use Existing IB Tables=0
UNET Froude Limit=0
UNET Froude Power=0
Write IC File=0
Echo Input=False
Echo Output=False
Write Detailed=0

--- RichCreek.f01 (steady flow) ---

Flow Title=NFF Regression Equation
Program Version=4.00
Number of Profiles=1
Profile Names=P100yr
River Rch & RM=RichCreek,Main      ,28246.3
909.3817
River Rch & RM=RichCreek,Main      ,25846.3
961.7458
River Rch & RM=RichCreek,Main      ,22531
1040.240
River Rch & RM=RichCreek,Main      ,21943.5
1049.816
Boundary for River Rch & Prof#=RichCreek,Main      ,1
Up Type=0
Dn Type=3
Dn Slope=0.016452

--- RichCreek.g01 (geometry) ---

Geom Title=USGS 3m DEM
Program Version=4.10

River Reach=RichCreek       ,Main
Reach XY= 30
     1938422.735      429985.453     1938650.822       430468.88
     1939118.915      430903.856     1939064.228       431220.82
      1939290.79      431825.731     1939741.515      432387.215
     1939703.985      433103.509     1939924.471      433525.553
     1939745.581      433995.625     1940022.108      435788.056
     1939143.221      437454.203     1938381.068      438070.523
     1937016.485      438603.509     1936499.124      439131.286
      1935500.86      439242.398     1935056.415      439487.189
     1933301.078      439239.682      1932032.11      439763.231
     1931426.967      440359.255     1930224.818       440589.62
     1929184.888        440348.3     1928242.179      441304.898
     1927681.415      441369.134      1927344.61      441610.453
     1927210.929      442428.161     1926733.499      443209.412
     1925591.138      443954.203     1924733.499      445542.745
     1924747.388      446207.676      1924402.14      446622.641

Type RM Length L Ch R = 1 ,28246.3 ,305.2,302.7,303.8
XS GIS Cut Line= 3
     1937963.938      430297.772     1938429.612      429992.713
     1938831.722      429626.164
#Sta/Elev= 30
       0 1277.11    39.8 1270.66    79.5 1266.46   149.1 1257.29   188.9 1250.11
   278.4  1225.3   367.8 1195.84   407.6    1186   437.4  1182.1   467.2 1181.74
   516.9  1183.3   549.2 1180.87   556.7 1180.44   564.2 1181.14   586.4 1183.95
   596.3 1186.12     626 1194.98   655.6 1208.27   675.4 1219.68   695.2 1233.04
     715 1248.04   774.3  1298.1   813.9 1329.72   863.4  1364.6   883.2 1377.26
     893 1381.55     903 1383.14   912.8 1382.85     992 1373.85  1100.8    1367
#Mann= 3 , 0 , 0
       0      .1       0   549.2    .045       0   564.2      .1       0
Bank Sta=549.2,564.2
XS Rating Curve= 0 ,0
Exp/Cntr=0.3,0.1

Type RM Length L Ch R = 1 ,27943.5 ,447.6,446.3,445.1
XS GIS Cut Line= 3
     1938119.255      430624.378     1938627.782      430205.617
     1938714.652      430054.595
#Sta/Elev= 30
       0  1345.8    39.9 1330.64    79.8 1317.08   119.8 1304.51   169.7 1289.72
   199.6 1279.92   219.6 1272.46   249.5 1259.93   279.5 1248.54   309.4 1235.99
   319.4 1232.67   339.4 1228.72   349.3 1226.16   389.3 1211.36   479.1 1177.14
   489.1 1174.52   499.1 1173.73     519 1174.04     539 1173.81     601 1172.02
   608.8 1171.87     616 1172.31   628.8 1174.14   668.4 1181.49   678.1 1183.33
   687.8 1185.85   726.5 1200.46   755.6 1212.34   794.3 1229.73     833 1248.24
#Mann= 3 , 0 , 0
       0      .1       0     601    .045       0     616      .1       0
Bank Sta=601,616
XS Rating Curve= 0 ,0
Exp/Cntr=0.3,0.1

Type RM Length L Ch R = 1 ,27497.4 ,229.9,231.3,233.1
XS GIS Cut Line= 4
     1938463.619      430819.502     1938733.363       430635.96
      1938935.17      430444.845     1939103.565      430404.751
#Sta/Elev= 30
       0 1320.07    29.7 1305.57    69.2 1286.98   168.1 1242.97     178 1238.25
   207.6 1223.45   227.4 1214.12   276.8 1192.01   326.3 1170.89   336.2 1167.46
   346.1 1165.96   405.7 1164.94   415.6 1164.53   439.9 1162.82   445.4 1162.52
   454.9 1162.67   465.2 1163.48   475.2 1164.73     495 1166.55   574.4 1172.49
   584.4 1173.82   594.3 1176.51   604.2 1179.67   642.7 1195.34   671.5 1207.97
   700.4 1221.43   719.6 1230.88   738.8 1241.01   748.5 1246.49   777.3 1264.48
#Mann= 3 , 0 , 0
       0      .1       0   439.9    .045       0   454.9      .1       0
Bank Sta=439.9,454.9
XS Rating Curve= 0 ,0
Exp/Cntr=0.3,0.1

Type RM Length L Ch R = 1 ,27265.7 ,231.9,235.3,238.4
XS GIS Cut Line= 3
     1938518.556      431083.347     1938989.194      430702.039
     1939410.871      430372.027
#Sta/Elev= 30
       0  1317.3    19.9 1313.93    39.7  1308.6   129.1 1278.22   198.6 1252.08
     288  1222.7   297.9 1218.54   307.8 1213.26   377.3  1172.3   387.3 1166.92
   397.2 1163.46   407.1 1162.62   446.8 1164.54   496.5 1163.86   536.2 1161.55
   575.9 1157.91   599.3 1157.22   605.7 1157.16   614.3 1157.51   655.3 1160.98
   665.2 1164.32   675.1 1169.55   724.7 1201.17   784.2 1241.18     814 1263.08
   873.4 1308.96   952.8 1364.84   972.6 1375.67  1032.1 1401.37  1141.2 1450.93
#Mann= 3 , 0 , 0
       0      .1       0   599.3    .045       0   614.3      .1       0
Bank Sta=599.3,614.3
XS Rating Curve= 0 ,0
Exp/Cntr=0.3,0.1

Type RM Length L Ch R = 1 ,27030.3 ,275.6,287.9,300.2
XS GIS Cut Line= 3
     1938710.643       431117.09     1938928.488      431008.836
     1939328.092      430774.953
#Sta/Elev= 30
       0 1247.29    68.1 1229.56   116.8  1215.6   136.2 1211.59   155.7 1209.49
   165.4 1206.66   175.2 1201.87   243.3 1163.49   253.1 1159.37     263 1157.85
   272.8 1157.64   351.6 1159.12   381.2 1158.73   410.7 1157.18   440.3 1154.03
   452.5 1153.43     460 1153.25   467.5 1153.37   469.8 1153.41   479.7 1154.82
   499.4 1159.53   509.2 1162.37   519.1 1166.51     529 1171.93   548.6 1184.87
   568.4 1196.89   588.1 1207.86   666.9 1250.55   686.6 1261.82   706.3 1273.63
#Mann= 3 , 0 , 0
       0      .1       0   452.5    .045       0   467.5      .1       0
Bank Sta=452.5,467.5
XS Rating Curve= 0 ,0
Exp/Cntr=0.3,0.1

Type RM Length L Ch R = 1 ,26742   ,273.1,263.6,254.7
XS GIS Cut Line= 4
      1938844.29      431221.334     1939020.704      431167.876
     1939279.913       431173.56     1939523.217      431076.996
#Sta/Elev= 30
       0 1267.52    29.1 1251.37    87.3 1214.63      97 1208.81   126.1 1192.65
   164.9 1168.81   174.6 1163.78   184.3 1159.56   204.3 1153.99   224.2 1149.94
     234 1148.88     249  1149.1     294 1151.25   413.7 1151.97   423.7  1152.6
   433.6 1154.55   443.6    1158   472.7 1171.44   521.2 1191.48   540.6 1199.91
   569.6 1213.92   608.4 1234.55   618.1 1240.15   627.8 1246.93   637.5 1255.69
   647.2 1265.12   656.9 1273.79   666.6 1281.24     686  1294.3   705.4 1306.49
#Mann= 3 , 0 , 0
       0      .1       0     234    .045       0     249      .1       0
Bank Sta=234,249
XS Rating Curve= 0 ,0
Exp/Cntr=0.3,0.1

Type RM Length L Ch R = 1 ,26478.2 ,306.5,309,310.7
XS GIS Cut Line= 3
     1938652.777      431610.373     1939158.104      431404.297
     1939677.337      431230.029
#Sta/Elev= 30
       0 1327.77    59.5 1307.35   119.1 1285.32   198.4  1262.8   267.9 1245.55
   317.5 1230.82     377 1217.02   416.7 1204.36   446.5 1197.13   456.4 1193.04
   466.4 1186.85   496.1 1166.05     506 1158.44     516 1149.55   525.9 1142.55
   527.8 1142.19   535.8 1140.66   542.8 1140.82   575.6 1142.62   635.4 1147.61
   675.2 1149.06     725 1149.29   734.9 1150.06   744.9 1152.04   774.8 1160.24
   864.4 1186.83   904.2 1200.35   944.1 1208.75  1023.7 1231.69  1093.4 1250.28
#Mann= 3 , 0 , 0
       0      .1       0   527.8    .045       0   542.8      .1       0
Bank Sta=527.8,542.8
XS Rating Curve= 0 ,0
Exp/Cntr=0.3,0.1

Type RM Length L Ch R = 1 ,26169.3 ,330.3,322.9,315.6
XS GIS Cut Line= 2
     1938921.805      431792.007      1939548.61       431612.92
#Sta/Elev= 30
       0 1321.01     9.9 1315.02    39.5 1297.58    49.4 1291.58    59.3 1285.47
   108.6 1254.05   118.5 1248.16   128.4 1242.57     158 1226.88   177.8 1216.74
   217.3 1197.08   246.9  1182.7   306.2 1153.63   316.1 1148.55   325.9 1142.79
   335.8 1137.21     339  1136.2   345.7 1134.07     354 1133.78   355.6 1133.72
   375.3 1134.81   395.1 1136.42   434.6 1139.89   444.5 1140.88   454.4 1142.44
   464.2 1144.68   474.1 1147.23   553.1 1169.54   622.3 1190.94   651.9 1200.74
#Mann= 3 , 0 , 0
       0      .1       0     339    .045       0     354      .1       0
Bank Sta=339,354
XS Rating Curve= 0 ,0
Exp/Cntr=0.3,0.1

Type RM Length L Ch R = 1 ,25846.3 ,272.3,271.2,270
XS GIS Cut Line= 3
     1938957.439      432282.469     1939407.671      431973.589
     1939857.903      431664.708
#Sta/Elev= 30
       0 1378.35    39.7 1369.66    69.5 1364.33    79.4 1361.75    99.3 1354.16
     129 1340.64   168.8 1323.67   188.6 1314.39   208.5 1304.12   327.6 1238.93
   496.4 1150.88   506.3  1145.6   526.2 1133.22   536.1 1129.79   538.5 1129.58
     546 1128.94   553.5 1129.03   575.8 1130.15   635.4 1135.45   704.8    1154
   804.1 1177.69   833.9 1186.23   863.7 1196.58   893.4 1208.57   923.2 1221.71
   943.1 1231.51     963 1242.32   982.8 1254.16  1012.6 1273.73    1092 1329.64
#Mann= 3 , 0 , 0
       0      .1       0   538.5    .045       0   553.5      .1       0
Bank Sta=538.5,553.5
XS Rating Curve= 0 ,0
Exp/Cntr=0.3,0.1

Type RM Length L Ch R = 1 ,25575.1 ,319.3,335.9,352.5
XS GIS Cut Line= 2
     1939138.436      432520.309     1940007.134      431856.159
#Sta/Elev= 30
       0  1295.6    69.6 1267.76    89.5 1259.02   119.3 1242.22   149.1 1221.66
     159 1215.82     169 1211.69   188.9 1208.66   208.8 1207.31   288.3 1208.05
     328 1204.89     338 1203.37   347.9 1200.52   397.6 1179.22     507 1138.01
   526.9 1128.83   536.8 1125.52   539.9 1125.28   546.8 1124.74   554.9 1125.14
   646.2 1130.36   695.9  1140.9   725.7 1150.77   755.5 1163.98     845 1211.96
   914.6 1246.35   994.1 1287.57  1053.7 1316.82  1073.6 1327.65  1093.5 1340.36
#Mann= 3 , 0 , 0
       0      .1       0   539.9    .045       0   554.9      .1       0
Bank Sta=539.9,554.9
XS Rating Curve= 0 ,0
Exp/Cntr=0.3,0.1

Type RM Length L Ch R = 1 ,25239   ,341.9,340.6,338.2
XS GIS Cut Line= 2
     1939443.029      432432.177     1940275.757      432502.914
#Sta/Elev= 30
       0 1181.82      10 1178.75    29.8  1172.3    39.8 1169.58    49.8 1167.31
    69.6 1164.06    79.6 1162.26    89.5 1160.04   238.8 1124.38   248.7 1122.43
   278.6 1117.75   287.5 1116.77   298.5 1116.37   302.5 1116.39   338.3 1116.72
   348.2  1118.2   358.2 1121.97   368.1 1127.28   407.9 1149.91   487.5 1194.83
   507.4 1205.84   527.3 1216.61     587 1247.92   626.8 1267.84   646.7 1278.27
   706.4 1311.22   716.3 1316.57   756.1 1337.49   795.9    1358   835.7 1378.11
#Mann= 3 , 0 , 0
       0      .1       0   287.5    .045       0   302.5      .1       0
Bank Sta=287.5,302.5
XS Rating Curve= 0 ,0
Exp/Cntr=0.3,0.1

Type RM Length L Ch R = 1 ,24898.3 ,371.8,369,367.4
XS GIS Cut Line= 3
     1939196.694      432778.013     1939753.553      432792.282
     1940263.622      432779.659
#Sta/Elev= 30
       0  1255.8   169.1 1194.05   318.3  1146.5   328.3  1145.2   338.2 1146.34
   358.1 1150.97     368 1151.04     378 1148.63   417.8 1136.33   487.4 1117.67
   507.3 1114.58   550.8 1110.83     557  1110.7   565.8 1111.81     577 1115.78
   607.1 1132.36   617.1  1138.6   687.1 1188.08   727.1 1215.35   757.1 1234.31
   787.1 1251.38   817.2 1266.41   837.2 1274.39   857.2 1279.07   887.2 1282.08
   897.2 1283.87   907.2 1287.16   917.2 1291.76   947.2 1307.72  1067.3 1374.88
#Mann= 3 , 0 , 0
       0      .1       0   550.8    .045       0   565.8      .1       0
Bank Sta=550.8,565.8
XS Rating Curve= 0 ,0
Exp/Cntr=0.3,0.1

Type RM Length L Ch R = 1 ,24529.2 ,188.4,183,176.9
XS GIS Cut Line= 3
      1939173.69      433200.776     1939766.455      433137.834
      1940184.77      433072.347
#Sta/Elev= 30
       0 1279.47    19.9 1278.25    49.7 1274.95   168.9  1259.7   198.7 1253.92
   258.3 1236.44   278.2 1228.89   288.1  1224.1     308 1213.23   337.8  1195.3
   367.6 1179.06   407.3 1159.21   447.1  1140.9   506.7 1110.76   516.6 1107.19
   526.6 1105.39   540.8 1104.45   546.4 1104.22   555.8  1104.5   625.6 1113.28
   645.3 1116.94     665 1121.87   674.9  1125.6   714.3 1143.64     734 1150.64
   802.9 1172.51   871.8 1199.05     921 1222.18   980.1  1248.6  1019.5 1269.05
#Mann= 3 , 0 , 0
       0      .1       0   540.8    .045       0   555.8      .1       0
Bank Sta=540.8,555.8
XS Rating Curve= 0 ,0
Exp/Cntr=0.3,0.1

Type RM Length L Ch R = 1 ,24346.3 ,459.7,471,482.9
XS GIS Cut Line= 3
     1939272.325      433491.649     1939804.975      433300.687
     1940159.377      433163.227
#Sta/Elev= 30
       0 1343.07    29.8 1326.41    69.5 1301.96    79.4 1296.27    99.3 1285.66
   158.8  1256.4   307.7 1184.58   337.5 1169.43   387.2 1143.31   397.1  1138.6
     407 1134.42   456.6 1115.06   476.5    1108   486.4 1105.02   496.4 1103.16
   506.3 1102.41   555.9 1101.27   558.3 1101.28   565.8 1101.32   573.3  1102.5
   575.8  1102.9   595.9 1110.24   615.9 1116.65   705.9 1142.84   725.9 1149.47
   765.9  1164.4   805.9 1181.02     876 1213.24     906 1228.15     946 1248.91
#Mann= 3 , 0 , 0
       0      .1       0   558.3    .045       0   573.3      .1       0
Bank Sta=558.3,573.3
XS Rating Curve= 0 ,0
Exp/Cntr=0.3,0.1

Type RM Length L Ch R = 1 ,23874.9 ,329.6,321.8,314.7
XS GIS Cut Line= 3
     1939295.327      433570.688     1939892.083      433716.525
     1940389.403      433817.331
#Sta/Elev= 30
       0 1312.78    39.6 1285.04    69.4  1265.4   148.6 1217.38   198.2 1190.18
   317.1 1130.55   336.9  1123.2   376.5 1110.96   426.1 1098.07   445.9 1096.06
   525.1 1092.85   525.3 1092.85   540.3 1093.71   584.6 1101.81   604.4 1107.68
   614.3 1113.03   634.2 1127.35   644.2 1133.46     674 1147.59   713.8 1164.07
   763.6 1179.93     883 1212.89   972.5 1235.12   992.4  1235.6  1032.2 1230.64
  1042.2 1230.25  1052.1 1231.45    1062 1234.51    1072 1239.07  1121.8  1265.3
#Mann= 3 , 0 , 0
       0      .1       0   525.3    .045       0   540.3      .1       0
Bank Sta=525.3,540.3
XS Rating Curve= 0 ,0
Exp/Cntr=0.3,0.1

Type RM Length L Ch R = 1 ,23553.2 ,340.1,335.5,330.2
XS GIS Cut Line= 3
     1939207.269      434119.958     1939738.033       434005.94
     1940295.669      433923.318
#Sta/Elev= 30
       0 1273.23    39.5 1254.91   118.4 1230.62   148.1 1216.84   197.4 1205.96
     227 1195.75   256.6 1183.11   325.7 1146.41   355.3 1132.18   375.1 1123.91
   404.7 1115.64   483.6 1089.06   493.5 1087.87   544.9 1086.84   559.9 1086.41
   562.6 1086.35   572.5 1087.38   582.4 1090.41   691.2 1135.78   720.9 1145.46
   750.6 1152.27   770.3 1155.11     800 1157.46   839.6  1158.1   859.4  1160.4
   869.2  1162.7   908.8 1178.15   948.4 1195.34  1037.4 1227.94  1106.6 1255.67
#Mann= 3 , 0 , 0
       0      .1       0   544.9    .045       0   559.9      .1       0
Bank Sta=544.9,559.9
XS Rating Curve= 0 ,0
Exp/Cntr=0.3,0.1

Type RM Length L Ch R = 1 ,23217.5 ,368.6,379.7,390.1
XS GIS Cut Line= 3
     1939341.029      434532.996     1939857.335      434319.274
     1940360.713      434125.478
#Sta/Elev= 30
       0 1259.84    29.9 1246.58    49.9 1238.87    89.8 1227.12   149.7 1212.15
   209.6 1195.29   259.4 1187.12   279.4 1182.24   369.2 1145.34   379.2 1139.81
   409.1 1116.65   419.1 1110.52   429.1 1106.17   528.9 1078.21   541.1 1076.09
   548.8 1075.62   556.1  1076.1   668.7 1091.27   698.6 1097.39   718.6 1103.11
   728.6 1106.84   778.6 1127.82   808.5 1141.81   878.4 1181.96   908.4 1197.72
   938.4    1211   988.3 1229.76  1018.3 1243.24  1048.2 1258.87  1098.2 1287.83
#Mann= 3 , 0 , 0
       0      .1       0   541.1    .045       0   556.1      .1       0
Bank Sta=541.1,556.1
XS Rating Curve= 0 ,0
Exp/Cntr=0.3,0.1

Type RM Length L Ch R = 1 ,22837.7 ,310,306.7,304.6
XS GIS Cut Line= 3
     1939343.782      434624.688     1939888.074      434680.121
     1940440.613      434725.038
#Sta/Elev= 30
       0 1292.61    19.9 1288.68    39.8  1283.2    99.5 1263.61   129.3 1252.49
     189 1227.58   208.9 1218.64   358.1 1141.35   407.8 1118.02   437.7 1103.24
   457.6 1094.98   507.3 1076.56   527.2 1070.92   536.9 1069.27   547.1 1069.06
   551.9 1069.86   586.7 1077.22   685.7 1093.75   774.8 1111.88   834.2 1124.82
   863.9 1141.62   873.8 1145.64   913.4 1158.12     953  1173.7   962.9 1178.54
   992.6 1196.36  1002.5 1201.62  1042.1 1220.16  1061.9  1227.2  1101.5 1237.85
#Mann= 3 , 0 , 0
       0      .1       0   536.9    .045       0   551.9      .1       0
Bank Sta=536.9,551.9
XS Rating Curve= 0 ,0
Exp/Cntr=0.3,0.1

Type RM Length L Ch R = 1 ,22531   ,302.3,301.2,299.5
XS GIS Cut Line= 3
     1939372.092      435008.523     1939917.803      434983.241
     1940463.678      434974.293
#Sta/Elev= 30
       0 1279.64    49.7  1260.6    99.3 1234.88   139.1 1218.76   178.8 1198.34
   208.6 1178.21     298 1106.52   327.8  1086.2   347.6 1075.91   357.6 1074.18
   417.2  1072.4   427.1 1075.97     437 1081.92     447 1085.12   456.9 1083.78
   506.6 1067.21   538.8 1062.71   546.3  1062.7   553.8 1064.69   615.8  1097.9
   655.5 1122.13     725 1168.73   814.3 1232.34   873.9 1271.07     993 1325.77
  1012.8 1338.46  1042.6 1360.19  1052.5 1364.99  1072.4 1366.36  1092.2 1363.72
#Mann= 3 , 0 , 0
       0      .1       0   538.8    .045       0   553.8      .1       0
Bank Sta=538.8,553.8
XS Rating Curve= 0 ,0
Exp/Cntr=0.3,0.1

Type RM Length L Ch R = 1 ,22229.7 ,289.7,286.2,282.8
XS GIS Cut Line= 3
      1939389.57      435296.234     1939902.775      435286.879
     1940477.341      435232.342
#Sta/Elev= 30
       0 1246.07   197.4 1154.81   217.2 1143.66   296.1 1094.12     306 1088.68
   325.7 1080.12   345.5 1074.75   414.6 1071.58   434.3 1072.24   454.1 1076.48
   463.9 1077.24   473.8 1075.18   513.3 1060.13   523.2 1058.45   536.9 1057.86
   543.1 1057.67   551.9 1058.08     563 1060.57     573 1064.58   602.8 1084.23
   622.8 1095.21   642.6 1108.53   712.3 1158.27   791.9 1210.16   831.7 1234.96
   911.3 1281.31   990.9 1338.48  1010.8 1348.56  1050.6 1365.84  1090.4 1379.13
#Mann= 3 , 0 , 0
       0      .1       0   536.9    .045       0   551.9      .1       0
Bank Sta=536.9,551.9
XS Rating Curve= 0 ,0
Exp/Cntr=0.3,0.1

Type RM Length L Ch R = 1 ,21943.5 ,356,370.1,385.9
XS GIS Cut Line= 3
      1939435.01      435606.295     1939851.989       435596.94
     1940499.231      435433.232
#Sta/Elev= 30
       0 1213.38    59.6 1197.34   109.2 1178.91   129.1 1172.88   278.1 1138.46
   307.8 1129.87   327.7 1121.56   357.5 1106.58   387.3 1089.63   407.2 1075.68
   417.1 1069.74     427 1068.14     447 1069.67   456.9 1069.39   466.9  1067.2
   506.8 1054.03   516.7 1051.96   526.4 1051.25   526.7 1051.23   541.4 1052.04
   636.3 1067.93   656.2 1073.48   676.2 1081.83   686.1 1086.89   765.8 1134.57
   835.6 1171.98   905.4 1214.58   925.3 1224.85   955.2 1238.41  1084.7 1306.43
#Mann= 3 , 0 , 0
       0      .1       0   526.4    .045       0   541.4      .1       0
Bank Sta=526.4,541.4
XS Rating Curve= 0 ,0
Exp/Cntr=0.3,0.1

Type RM Length L Ch R = 1 ,21573.4 ,492.2,496,498
XS GIS Cut Line= 3
      1939525.89      435746.625     1939949.551      435907.001
     1940444.665      436147.576
#Sta/Elev= 30
       0 1220.72    19.7 1211.49    88.6 1171.38   147.7 1139.96   206.8 1111.91
   275.7 1081.78     325  1057.3   334.8 1054.89   344.7 1054.09   393.9 1052.46
   423.5 1050.52   449.3 1045.27     453 1044.42   464.3 1046.08     483 1053.45
     513 1061.29   523.1 1066.26   583.1 1105.01   633.2 1138.79   683.2 1168.16
   723.2 1189.41   773.3 1212.58   803.3 1224.04   833.3    1233   853.3 1241.82
   903.4 1268.11   943.4 1286.94   973.4 1304.91   993.5 1318.32  1003.5 1325.85
#Mann= 3 , 0 , 0
       0      .1       0   449.3    .045       0   464.3      .1       0
Bank Sta=449.3,464.3
XS Rating Curve= 0 ,0
Exp/Cntr=0.3,0.1

Type RM Length L Ch R = 1 ,21077.4 ,289.1,288.5,287.8
XS GIS Cut Line= 3
     1939326.868      436099.596     1939799.232      436382.046
     1940257.622      436677.209
#Sta/Elev= 30
       0  1224.3      70 1184.65   140.1 1139.63   170.1 1122.08   240.2  1085.2
   280.2 1066.31   300.2 1058.24   330.2 1047.68   340.2 1045.05   350.2  1043.7
   390.3  1041.3   500.3 1038.44   505.4 1038.45   520.4 1040.05   530.4 1045.13
   540.4 1052.34   560.3 1064.35   599.9 1083.76   649.5 1110.09   689.2 1127.77
   748.6 1149.96   768.4  1159.3   798.2 1175.31   847.8 1198.75   877.5 1215.54
   917.1 1236.23     937  1247.9  1036.1 1313.66  1075.7 1338.78  1095.6 1350.47
#Mann= 3 , 0 , 0
       0      .1       0   505.4    .045       0   520.4      .1       0
#XS Ineff= 2 , 0
          411.59 1054.74
Permanent Ineff=
       F       F
Bank Sta=505.4,520.4
XS Rating Curve= 0 ,0
Exp/Cntr=0.3,0.1

Type RM Length L Ch R = 1 ,20788.6 ,284.3,278,271.8
XS GIS Cut Line= 2
     1939189.099      436358.728     1940041.768      436845.204
#Sta/Elev= 30
       0 1242.79      30 1219.14    70.1  1185.3    90.2 1170.26   150.3  1129.8
   170.3 1118.29   190.3 1108.44   210.4 1099.47   290.5 1070.53   330.6 1054.04
   350.6 1043.93   360.6 1040.79   370.6 1038.84   410.7 1036.76   448.5  1032.5
   450.8 1032.33   463.5 1034.03   500.9 1041.28   510.9 1045.69   550.9 1066.94
     601 1088.64   661.1  1116.7   711.2  1138.1   761.3 1157.35   791.4 1166.75
   891.5 1194.58   901.6 1196.42   941.6 1198.02   961.6  1202.7   981.7 1209.22
#Mann= 3 , 0 , 0
       0      .1       0   448.5    .045       0   463.5      .1       0
Bank Sta=448.5,463.5
XS Rating Curve= 0 ,0
Exp/Cntr=0.3,0.1

Type RM Length L Ch R = 1 ,20510.8 ,371.8,379.7,387.7
XS GIS Cut Line= 2
     1939158.361      436754.324     1939948.215      436942.766
#Sta/Elev= 30
       0 1175.94    19.8 1166.08    49.5  1149.1      99 1124.64   138.6 1103.65
   168.4 1086.67   227.8 1051.02   247.6  1039.9   257.5 1036.04   267.4 1033.99
     307  1028.3   312.9 1027.84   326.8 1027.41   327.9 1027.45   396.1 1031.76
   445.6 1032.67   455.5 1033.86   465.4  1036.5   495.1 1045.58   514.9 1052.36
   564.4 1072.11   604.1 1086.61   673.4 1109.38   693.2 1115.04     713 1122.54
   732.8 1127.74   752.6 1136.72   762.5 1142.04   792.2 1159.51     812 1169.21
#Mann= 3 , 0 , 0
       0      .1       0   312.9    .045       0   327.9      .1       0
Bank Sta=312.9,327.9
XS Rating Curve= 0 ,0
Exp/Cntr=0.3,0.1

Type RM Length L Ch R = 1 ,20131   ,251.5,253.4,255.3
XS GIS Cut Line= 3
      1939060.56      436994.565     1939325.551      437169.925
     1939780.878      437471.244
#Sta/Elev= 30
       0 1139.03    29.8  1123.3   109.2 1080.28     139 1064.68   198.6 1034.21
   208.5 1030.58   218.5 1028.93   248.2 1027.32   310.3 1021.72   317.8 1021.31
   325.3 1021.26   327.7 1021.24   387.2 1023.26   397.2 1023.94   407.1  1026.4
     417 1030.58   446.8 1045.74   496.4 1072.07   516.3 1082.98   536.2 1094.54
     556 1106.78   575.9 1119.62   635.4 1159.48   655.3 1172.25   675.1 1184.45
     695 1196.08   714.8 1206.74   764.5 1232.33   784.3 1241.78   863.8 1278.21
#Mann= 3 , 0 , 0
       0      .1       0   310.3    .045       0   325.3      .1       0
Bank Sta=310.3,325.3
XS Rating Curve= 0 ,0
Exp/Cntr=0.3,0.1

Type RM Length L Ch R = 1 ,19877.6 ,341,346.6,352.2
XS GIS Cut Line= 2
     1938888.394      437145.909     1939619.945      437722.976
#Sta/Elev= 30
       0 1136.54    99.1 1098.63   188.3 1061.46   218.1 1050.65   267.6  1034.2
   277.6 1031.31   287.5 1029.19   376.3 1019.26   386.6 1018.87   391.3 1019.01
   406.4 1019.72   416.3 1020.95   426.2 1023.68     446 1032.16   465.9 1042.48
   495.6 1059.86   525.4 1079.16   555.1 1100.16   604.6 1136.86   644.3 1164.06
   664.1 1175.84   713.7 1200.54   723.6 1204.59   733.5 1207.03   743.4  1208.7
   783.1 1222.84   802.9 1229.13   882.2 1250.83   892.1 1254.19   931.8 1270.03
#Mann= 3 , 0 , 0
       0      .1       0   376.3    .045       0   391.3      .1       0
Bank Sta=376.3,391.3
XS Rating Curve= 0 ,0
Exp/Cntr=0.3,0.1

Type RM Length L Ch R = 1 ,19531   ,308.5,306.1,303.6
XS GIS Cut Line= 2
     1938618.264      437198.412     1939284.069      438063.957
#Sta/Elev= 30
       0 1187.29    59.6 1178.06    89.4  1170.9   119.1 1162.76     139 1155.95
   188.6 1135.55     278  1105.3   297.8 1097.49   307.8 1092.52   347.4 1071.03
     407 1041.25     417 1035.53   436.8 1021.94   446.7 1018.45   456.6  1017.5
   538.5 1013.81   553.5 1013.39   575.8 1012.64   585.7 1013.12   595.6 1016.12
   625.4 1033.22   724.7 1086.99     824  1139.6   873.6 1164.96     963 1212.12
   982.8 1221.76  1012.6 1232.78  1032.4 1241.15  1052.3 1251.04    1092 1272.95
#Mann= 3 , 0 , 0
       0      .1       0   538.5    .045       0   553.5      .1       0
Bank Sta=538.5,553.5
XS Rating Curve= 0 ,0
Exp/Cntr=0.3,0.1

Type RM Length L Ch R = 1 ,19224.9 ,316.9,327.8,338.8
XS GIS Cut Line= 3
     1938518.191      437688.517     1938647.829       437755.34
     1939096.523      438223.877
#Sta/Elev= 30
       0  1102.1    58.3  1062.9    77.8 1051.55    97.2 1041.09   116.7 1031.44
   145.8 1019.25   155.8 1015.72   165.8 1013.05   175.8 1011.73   215.7 1009.95
   241.4 1008.23   245.6 1007.96   256.4 1008.16   305.5 1011.59   315.5 1013.19
   325.5 1016.36   385.4  1043.6   405.3 1053.77   425.3 1065.56   465.2  1093.3
   485.2 1104.43   495.2  1109.3   525.1 1121.27     585 1147.06   624.9 1163.44
   654.8 1176.26   674.8 1186.04   714.7 1208.05   734.7  1217.4   794.6 1243.97
#Mann= 3 , 0 , 0
       0      .1       0   241.4    .045       0   256.4      .1       0
Bank Sta=241.4,256.4
XS Rating Curve= 0 ,0
Exp/Cntr=0.3,0.1

Type RM Length L Ch R = 1 ,18897   ,186.1,188.3,190.3
XS GIS Cut Line= 3
      1938392.34      437840.874     1938435.107      437949.574
     1938558.062      438373.681
#Sta/Elev= 30
       0 1083.64    19.5 1071.46    48.7 1052.72    97.3 1020.67   107.1 1014.68
   116.8 1010.09   126.6 1007.39   136.4 1005.96   165.9 1002.93   185.5 1000.32
   189.7 1000.15   195.3  999.92   204.7 1000.39   224.8 1002.03   254.2 1003.98
     264 1005.51   273.8 1008.48   283.6 1012.56   322.9 1029.67   352.3 1041.88
   371.9 1050.28   391.6 1059.08     421 1072.62   430.8 1077.29   450.4 1086.85
   470.1 1096.82   509.3 1117.42   519.1 1122.72   538.8 1133.67   558.4 1145.26
#Mann= 3 , 0 , 0
       0      .1       0   189.7    .045       0   204.7      .1       0
Bank Sta=189.7,204.7
XS Rating Curve= 0 ,0
Exp/Cntr=0.3,0.1

Type RM Length L Ch R = 1 ,18708.8 ,503,485.4,468
XS GIS Cut Line= 3
     1938187.448      437574.201     1938287.315       438110.98
     1938394.301      438646.455
#Sta/Elev= 30
       0 1228.26    29.8 1217.08    89.3 1191.26     139 1163.07   188.6 1132.42
   198.5 1127.29   238.2 1109.03   287.9 1084.52   347.4  1045.6   377.2 1030.63
     407 1018.43   436.8 1009.51   476.5 1001.09   525.9  993.06   536.1  993.15
   540.9  994.13     546  995.17   565.8 1002.28   595.6 1016.67   625.4  1033.5
   665.1 1058.59     685 1070.04     814 1139.24   863.7 1163.98     963    1224
   982.8 1237.24  1012.6 1259.03  1022.6 1265.04  1052.3 1280.45    1092 1298.33
#Mann= 3 , 0 , 0
       0      .1       0   525.9    .045       0   540.9      .1       0
Bank Sta=525.9,540.9
XS Rating Curve= 0 ,0
Exp/Cntr=0.3,0.1

Type RM Length L Ch R = 1 ,18222.7 ,227.7,242.5,257.3
XS GIS Cut Line= 2
     1937579.766      438085.003     1938092.971      438462.779
#Sta/Elev= 30
       0 1066.41    99.6 1038.07   109.5 1034.82   119.5 1030.82   129.4  1025.3
   139.4 1018.52   159.3 1003.43   169.3  997.57   179.2  994.06   189.2  992.19
   199.1  991.13     229  989.35   248.9  988.89   288.8  988.68   317.8  988.06
   328.6  987.98   332.8     988   358.5  988.14   368.4  989.34   378.4  992.54
   418.2 1011.96   438.1 1022.23   448.1 1027.75     468 1039.37   497.9 1057.49
   537.7 1082.21   547.6 1087.89   557.6 1093.24   607.4 1118.23   637.2 1132.52
#Mann= 3 , 0 , 0
       0      .1       0   317.8    .045       0   332.8      .1       0
#XS Ineff= 2 , 0
          244.09 1012.34
Permanent Ineff=
       F       F
Bank Sta=317.8,332.8
XS Rating Curve= 0 ,0
Exp/Cntr=0.3,0.1

Type RM Length L Ch R = 1 ,17980.9 ,250.1,249.8,249.5
XS GIS Cut Line= 3
     1937519.179      438190.139     1937608.277      438325.568
     1937772.218      438836.991
#Sta/Elev= 30
       0 1081.09    28.6  1066.4    47.7 1055.68    76.3 1038.92    85.8 1032.61
    95.4 1024.96   114.4 1007.72     124 1000.24   133.5  994.78     143  991.47
   152.6  990.23   201.9  987.67   228.8  985.65   243.8  985.06   261.6  984.56
   301.4  982.71   351.1  982.94     361  983.39     371  985.49   380.9  989.68
   390.9  994.52   410.8 1002.15   420.7 1007.32   470.4 1040.44   559.9 1096.08
   569.9  1101.7   609.7 1122.94   649.4 1145.55   679.3    1162   699.2  1173.7
#Mann= 3 , 0 , 0
       0      .1       0   228.8    .045       0   243.8      .1       0
Bank Sta=228.8,243.8
XS Rating Curve= 0 ,0
Exp/Cntr=0.3,0.1

Type RM Length L Ch R = 1 ,17731   ,186.5,189.8,193
XS GIS Cut Line= 3
     1937222.295      437954.741     1937394.956      438472.722
     1937567.616      438990.703
#Sta/Elev= 30
       0 1153.62    49.6 1142.61    89.4    1135     139 1123.08   168.8 1114.45
   228.3 1094.73   248.2 1086.37   337.5 1045.15   357.4 1035.36     407  1009.7
     417 1003.86   436.8  989.46   446.7  983.44   456.6  980.66   496.4  977.81
   538.5  976.02     546  975.88   553.5  976.11   595.6  978.75   645.3  980.76
   655.2  982.16   665.1  985.92     675  991.68     685  998.46   734.6 1034.72
   764.4 1057.58   774.3 1063.92     953 1161.55  1032.4 1203.64    1092 1234.34
#Mann= 3 , 0 , 0
       0      .1       0   538.5    .045       0   553.5      .1       0
Bank Sta=538.5,553.5
XS Rating Curve= 0 ,0
Exp/Cntr=0.3,0.1

Type RM Length L Ch R = 1 ,17541   ,477.5,463.7,450
XS GIS Cut Line= 3
     1937182.908       438355.75     1937229.239       438610.57
     1937464.943      439063.941
#Sta/Elev= 30
       0  998.74    19.9  994.86    39.8  991.69   139.5  978.01   174.4  972.04
   179.3  971.37   189.3  971.06   189.4  971.06   219.2  972.78   239.1  975.02
     249  976.86     259  980.17   268.8  985.27   278.6   991.2   288.5  996.49
   327.8 1019.36   357.3 1034.61   376.9 1045.76   396.6 1058.26     426 1078.65
   445.7 1091.56   465.4 1102.95     485 1113.26   504.7 1122.58   524.3 1130.94
   573.4 1148.33   593.1  1155.9   612.8 1164.72   661.9 1187.82     770 1237.08
#Mann= 3 , 0 , 0
       0      .1       0   174.4    .045       0   189.4      .1       0
Bank Sta=174.4,189.4
XS Rating Curve= 0 ,0
Exp/Cntr=0.3,0.1

Type RM Length L Ch R = 1 ,17077.5 ,246.3,249.7,253.2
XS GIS Cut Line= 3
     1936669.184      438683.742     1936804.613      438747.892
     1937226.938      439168.435
#Sta/Elev= 30
       0 1082.56      10 1079.41      20 1074.66      30 1068.52      50 1054.21
    69.9 1037.34   109.9 1000.46   119.9  992.35   129.9  985.38   139.9  979.37
   159.8  968.68   169.7  964.54   177.1  963.07   189.6  962.44   192.1  962.61
   259.1  968.07   308.8  969.25   318.7  970.27   328.6  972.14   338.6  975.12
   348.5  979.43   358.4  985.37   368.4  992.26   388.2 1007.46   398.2 1013.73
   447.8 1040.26   497.5 1068.84     577 1112.47   626.6  1136.4   745.8 1191.16
#Mann= 3 , 0 , 0
       0      .1       0   177.1    .045       0   192.1      .1       0
Bank Sta=177.1,192.1
XS Rating Curve= 0 ,0
Exp/Cntr=0.3,0.1

Type RM Length L Ch R = 1 ,16827.8 ,349.1,356.5,364
XS GIS Cut Line= 3
     1936628.199      438769.276     1936642.454      438904.705
     1936956.079       439318.12
#Sta/Elev= 30
       0 1045.69    38.9 1023.68    48.6 1017.66    87.5  989.38    97.3  983.47
     107   978.5   116.7  974.49   136.2  968.93   166.1   963.9     196  961.22
   230.9  960.04     236  959.99   245.9  960.59   265.9   963.8   275.9  964.71
   315.8  964.71   325.8  965.04   335.8  966.18   345.7  968.05   355.7  970.68
   365.7  975.01   375.7  981.57   395.6  997.08   425.6 1017.54   455.5 1039.68
   465.5 1046.46   495.4 1063.54   555.3 1096.14   625.2 1132.97   655.1 1149.27
#Mann= 3 , 0 , 0
       0      .1       0   230.9    .045       0   245.9      .1       0
Bank Sta=230.9,245.9
XS Rating Curve= 0 ,0
Exp/Cntr=0.3,0.1

Type RM Length L Ch R = 1 ,16471.1 ,236,240.1,241.8
XS GIS Cut Line= 2
     1936328.829      438920.743     1936567.312      439672.099
#Sta/Elev= 30
       0 1006.41    29.9  990.02    39.9  985.57    59.9  978.78    79.8  973.01
    89.8  970.58   109.8  966.76   129.7  963.98   199.6  957.37   234.6  953.56
   239.5  953.16   249.5  953.15   249.6  953.16   269.4  954.61   279.4  956.23
   309.3  963.18   329.3  968.53   339.3  971.74   369.2  982.97   389.2  991.85
   399.1  996.88     459 1030.55     469 1035.72   488.9 1045.16   538.8 1066.96
   698.5 1133.77   738.4 1152.03   748.4 1157.03   758.4 1162.72   788.3 1182.19
#Mann= 3 , 0 , 0
       0      .1       0   234.6    .045       0   249.6      .1       0
Bank Sta=234.6,249.6
XS Rating Curve= 0 ,0
Exp/Cntr=0.3,0.1

Type RM Length L Ch R = 1 ,16231   ,318.2,320.1,324.5
XS GIS Cut Line= 3
     1936102.149      438665.444     1936169.715      439210.239
     1936296.781      439741.989
#Sta/Elev= 30
       0 1207.23      20 1200.53    39.9 1191.75   189.6 1117.34   249.5 1088.92
   299.4 1066.32   319.4 1056.42   359.3 1034.37   379.3 1022.46   389.3 1015.56
   399.2 1007.91   429.2   983.4   439.2  976.14   449.2  969.85   459.1  964.45
   469.1  960.16   479.1  957.21     509  953.51   541.5  948.66     549  948.46
   556.5  948.78   598.7  951.51   628.5  957.16   648.4     962   698.1  976.42
   737.8  989.99   787.5 1008.92   867.1 1041.69   986.4 1096.42  1095.7 1145.04
#Mann= 3 , 0 , 0
       0      .1       0   541.5    .045       0   556.5      .1       0
Bank Sta=541.5,556.5
XS Rating Curve= 0 ,0
Exp/Cntr=0.3,0.1

Type RM Length L Ch R = 1 ,15910.5 ,282.8,278.9,274.5
XS GIS Cut Line= 2
     1935844.136      439018.751     1935872.305      439757.148
#Sta/Elev= 30
       0 1033.11      20 1022.86    69.9  994.54   139.8  956.83   169.8  942.49
   179.7  938.83     185  937.89   189.7  937.05   199.7  936.88     200   936.9
   309.6  945.95   349.5  947.87   359.5  949.07   369.5  950.89   389.4   955.8
   409.4  961.95   419.4  965.73   429.4  970.15   439.4  975.45   449.4  981.49
   469.3   995.2   499.3 1017.11   509.3 1023.68   519.2 1029.17   549.2 1041.24
   559.2 1045.76   629.1 1081.02   649.1 1091.94     699  1122.3   738.9 1144.12
#Mann= 3 , 0 , 0
       0      .1       0     185    .045       0     200      .1       0
Bank Sta=185,200
XS Rating Curve= 0 ,0
Exp/Cntr=0.3,0.1

Type RM Length L Ch R = 1 ,15631.4 ,306,300,293.4
XS GIS Cut Line= 3
      1935461.71      438696.764     1935575.036      439232.811
     1935703.689      439763.874
#Sta/Elev= 30
       0  1144.8    19.9 1135.87    79.7  1107.1   109.6 1095.92   129.5 1090.94
   139.5 1087.69   149.4 1083.24   179.3 1067.77   278.9 1019.04   318.8  998.28
   388.5   968.5   448.3   946.6   468.2   940.5   488.1  937.32   540.4  933.15
   547.9  933.02   555.4  933.76   567.8  936.21   577.7  939.08   597.6  946.13
     677  986.23   726.7 1013.95   756.5 1028.24   776.4 1036.51   816.1 1050.25
   845.9 1059.47   885.7 1067.93   905.6 1072.99  1044.6 1112.01  1094.3 1124.69
#Mann= 3 , 0 , 0
       0      .1       0   540.4    .045       0   555.4      .1       0
Bank Sta=540.4,555.4
XS Rating Curve= 0 ,0
Exp/Cntr=0.3,0.1

Type RM Length L Ch R = 1 ,15331.4 ,288.9,300,312.6
XS GIS Cut Line= 3
     1935138.479      439018.751     1935288.376      439313.226
     1935571.345      439801.981
#Sta/Elev= 30
       0 1099.88      40 1080.36   130.2  1038.5   150.2 1027.94   160.2 1020.24
   170.2 1010.56   200.3  975.99   210.3  965.91   220.3  957.74   230.3  951.19
   240.3  946.24   260.3  939.67   280.4  936.44   322.9  931.41   337.9   930.6
   350.2  931.85   370.1  937.15   409.7  955.01   429.5  960.54   459.2  963.66
   518.7  967.13   528.6  969.05   538.5  974.37   548.4  983.28   558.3  993.63
   568.2 1002.66   578.1 1008.51   617.8 1021.67   786.2 1063.08   895.2 1085.89
#Mann= 3 , 0 , 0
       0      .1       0   322.9    .045       0   337.9      .1       0
Bank Sta=322.9,337.9
XS Rating Curve= 0 ,0
Exp/Cntr=0.3,0.1

Type RM Length L Ch R = 1 ,15031.4 ,335.6,338.4,342.6
XS GIS Cut Line= 3
     1935058.291      439211.202     1935053.023      439486.947
      1935035.64      440017.952
#Sta/Elev= 30
       0 1022.53     9.8 1017.87    39.4 1001.62    98.5  965.55   118.2  955.01
   137.9  946.16   147.8  942.89   167.4  939.32   226.6  931.65   256.1  927.19
     266  926.79   268.3  926.88   283.3  927.74   305.3  929.53   344.7  934.39
   354.5  936.85   364.3  940.74   374.2  946.22     384  953.15   393.9  960.99
   423.4  986.55   433.2  993.72   472.6  1019.3   492.2 1031.52     571 1078.21
   620.2 1105.21   649.7 1122.04     689 1143.18     748 1177.16   807.1 1209.42
#Mann= 3 , 0 , 0
       0      .1       0   268.3    .045       0   283.3      .1       0
Bank Sta=268.3,283.3
XS Rating Curve= 0 ,0
Exp/Cntr=0.3,0.1

Type RM Length L Ch R = 1 ,14692.6 ,261.1,261.2,259.7
XS GIS Cut Line= 3
     1934771.395      439134.578     1934737.538      439378.707
      1934616.22      439907.752
#Sta/Elev= 30
       0 1021.59    39.4 1006.53    49.3 1002.43    59.2  997.32    78.9  984.43
   118.3  956.44     138     945   147.9  940.57   157.7  937.32   167.6  935.27
   197.2  930.87   226.8  922.02   235.4  921.01   236.6  920.87   250.4  921.09
   285.9   923.2   295.8  924.15   305.7  926.25   325.4  933.39   345.2  941.76
   414.2   974.3     434  982.08   453.7  988.24   483.3     996   512.9 1002.48
   591.9 1015.02   690.6 1034.96   710.3 1039.54   769.5 1061.48   789.2 1069.63
#Mann= 3 , 0 , 0
       0      .1       0   235.4    .045       0   250.4      .1       0
Bank Sta=235.4,250.4
XS Rating Curve= 0 ,0
Exp/Cntr=0.3,0.1

Type RM Length L Ch R = 1 ,14431.4 ,299.5,300,300.5
XS GIS Cut Line= 3
      1934562.07      438774.996     1934484.855      439315.508
      1934407.64      439856.021
#Sta/Elev= 30
       0 1095.06    39.7  1081.4    99.3 1062.18   148.9 1043.97   188.6 1030.77
   218.4 1023.44     278 1012.49   307.8 1003.34   317.7   999.9   337.5  991.37
     407  955.46   426.9  946.56   456.6  936.12   486.4  926.56   538.5  915.65
     546  914.95   553.5  915.14   575.8   917.3   585.7   919.9   595.6  924.73
   704.8  991.07   774.3 1029.01   794.2 1038.94   853.8 1065.98   903.4 1089.96
   943.1 1110.79   982.8 1134.51   992.7 1139.62  1062.2 1171.57    1092 1183.32
#Mann= 3 , 0 , 0
       0      .1       0   538.5    .045       0   553.5      .1       0
Bank Sta=538.5,553.5
XS Rating Curve= 0 ,0
Exp/Cntr=0.3,0.1

Type RM Length L Ch R = 1 ,14131.4 ,304.7,300,295.3
XS GIS Cut Line= 3
     1934279.687      438723.185     1934189.924      439261.756
     1934100.162      439800.327
#Sta/Elev= 30
       0 1137.34    79.4 1099.98   148.9 1057.15   158.8 1052.85   198.6 1038.16
   287.9  997.84   367.3  964.78   466.6  926.18   486.4  920.31   538.5  911.27
     546  910.54   553.5  910.57   565.8  911.48   575.8  913.28   585.7   916.5
     675  960.96     685  965.18   694.9  967.91   734.6  973.01   754.5  972.13
   764.4  973.98   774.3  979.15   833.9 1023.83   863.7 1044.51   873.6 1050.34
   893.4 1058.48   943.1 1073.91   972.9 1084.26  1052.3 1115.69    1092 1129.84
#Mann= 3 , 0 , 0
       0      .1       0   538.5    .045       0   553.5      .1       0
Bank Sta=538.5,553.5
XS Rating Curve= 0 ,0
Exp/Cntr=0.3,0.1

Type RM Length L Ch R = 1 ,13831.4 ,298.5,300,301.6
XS GIS Cut Line= 3
     1933869.405      438684.467     1933892.784      439229.966
     1933916.163      439775.465
#Sta/Elev= 30
       0 1169.96   158.8  1082.5   208.5 1060.43     278  1032.2   337.5 1006.69
   357.4  996.38   397.1  972.83   496.4  918.95   516.2  911.93   538.5  906.63
     546  905.77   553.5  905.99   575.8  908.41   595.6  912.13   655.2  928.65
   665.1  930.35     685  928.94   694.9  929.41   704.8  932.46   714.8  937.44
   744.6  955.91   764.4   965.3   843.8 1006.01   853.8 1009.59   863.7 1011.32
   883.5 1012.85   893.4  1015.1   992.7 1058.87  1052.3 1079.74    1092 1096.33
#Mann= 3 , 0 , 0
       0      .1       0   538.5    .045       0   553.5      .1       0
Bank Sta=538.5,553.5
XS Rating Curve= 0 ,0
Exp/Cntr=0.3,0.1

Type RM Length L Ch R = 1 ,13531.4 ,304,300,295.3
XS GIS Cut Line= 3
      1933606.59       438694.59     1933593.065      439240.426
     1933577.903      439786.215
#Sta/Elev= 30
       0 1118.14    59.6  1091.5   129.1 1067.68   178.7 1044.35     278 1000.95
   397.1  955.27   476.5   914.7   486.4  910.95   496.4  908.46   526.2  902.67
   538.5  901.29     546  901.18   553.5   902.1   575.8  906.21   625.4  908.18
   635.4  909.76   655.2  915.14     685   927.3   734.6  945.74   794.2  978.16
     824  997.55   833.9 1001.22   873.6 1009.75   943.1 1019.61     963  1026.6
  1002.7 1043.92  1032.4  1054.4  1042.4 1057.18  1072.2 1062.54    1092 1068.41
#Mann= 3 , 0 , 0
       0      .1       0   538.5    .045       0   553.5      .1       0
Bank Sta=538.5,553.5
XS Rating Curve= 0 ,0
Exp/Cntr=0.3,0.1

Type RM Length L Ch R = 1 ,13231.4 ,618.8,613.9,609.5
XS GIS Cut Line= 3
     1933209.805      438703.076     1933293.264      439241.079
     1933394.107      439786.574
#Sta/Elev= 30
       0 1093.54    39.6 1085.37    79.2 1083.08    89.1 1081.28   178.2 1050.42
   207.9 1037.77   277.2 1001.36   336.6   979.8   405.8  943.46   435.6  929.67
   494.9  904.62   536.9  895.55   551.9   894.4   554.3  894.35   633.6  899.09
   653.4  898.75   663.3  900.16   673.2   904.1     693  916.28   811.9  998.42
   851.5 1030.27   861.4 1037.58   871.3 1043.19   891.2 1051.33   920.9 1057.66
   930.8 1061.78   960.5 1079.96   990.2 1091.84  1019.9 1105.64  1099.2 1136.68
#Mann= 3 , 0 , 0
       0      .1       0   536.9    .045       0   551.9      .1       0
Bank Sta=536.9,551.9
XS Rating Curve= 0 ,0
Exp/Cntr=0.3,0.1

Type RM Length L Ch R = 1 ,12617.4 ,294.2,294.1,294.1
XS GIS Cut Line= 2
     1932522.263       438939.75     1932831.137      439726.189
#Sta/Elev= 30
       0 1107.02     9.9 1103.64    49.7 1083.17    69.6 1075.38    99.4 1066.52
   139.2 1056.69     169 1047.29   178.9 1042.68   188.9 1035.07   208.7 1013.84
   228.6  997.26   268.4  969.18   318.1  936.19   347.9  913.97   357.8  908.34
   367.8  905.96   417.5  907.31   437.4  903.37   477.1  892.17   533.2  884.07
   536.8   883.8   548.2  883.97   646.1  892.32   656.1  892.52   695.8  889.86
   705.8  891.65   715.7  896.78   735.6   909.8   795.2  952.68   844.9  986.11
#Mann= 3 , 0 , 0
       0      .1       0   533.2    .045       0   548.2      .1       0
Bank Sta=533.2,548.2
XS Rating Curve= 0 ,0
Exp/Cntr=0.3,0.1

Type RM Length L Ch R = 1 ,12323.3 ,247.4,244.7,242
XS GIS Cut Line= 3
      1932325.06      439129.826     1932374.955      439367.421
     1932655.787      440075.118
#Sta/Elev= 30
       0 1060.77    29.1 1038.39    58.3 1012.95      68 1006.44   116.5  984.14
   155.4  962.81   194.2     938   242.8  900.64   252.7  896.32   262.6  895.66
   292.2  898.03   302.1  896.71   331.8  884.91   391.1  887.26   450.4  878.35
   450.7  878.35   465.7  878.99   539.4  889.62   569.1  889.19     579  890.62
   588.9  897.12   628.4  937.55   648.2  954.52     668  968.59   697.6  986.97
   717.4  995.36   776.7 1004.06   885.5 1012.24   915.2 1011.22  1004.2 1003.33
#Mann= 3 , 0 , 0
       0      .1       0   450.7    .045       0   465.7      .1       0
Bank Sta=450.7,465.7
XS Rating Curve= 0 ,0
Exp/Cntr=0.3,0.1

Type RM Length L Ch R = 1 ,12078.6 ,352.5,343.7,334.8
XS GIS Cut Line= 3
     1931961.992      439169.279     1932222.305      439649.231
     1932482.618      440129.182
#Sta/Elev= 30
       0 1053.69    99.3 1022.26     278  945.35   307.8  929.05   337.5  906.78
   347.4  900.61   357.4  896.28   367.3  893.58   377.2  892.23   426.9   889.5
   456.6  884.65   506.3  881.73   536.1  874.59     546  873.86   551.8  873.87
   566.8  874.31   655.2  880.55   665.1  882.08     675  886.05   694.9  898.96
   714.8  907.71   724.7  910.92   794.2  923.76     814  928.56   853.8  940.12
   873.6  947.88   923.2  970.26   972.9  989.03  1052.3 1022.04    1092 1036.42
#Mann= 3 , 0 , 0
       0      .1       0   551.8    .045       0   566.8      .1       0
Bank Sta=551.8,566.8
XS Rating Curve= 0 ,0
Exp/Cntr=0.3,0.1

Type RM Length L Ch R = 1 ,11734.8 ,266.2,266.4,266.5
XS GIS Cut Line= 3
     1931707.313      439688.174      1931873.63       439790.34
     1932341.691      440170.491
#Sta/Elev= 30
       0  993.34    58.6  954.74    87.8  935.19    97.6  929.05   107.4   923.5
   126.9  913.34   165.9  894.26   195.2  881.47   205.1  877.59     215  874.41
   224.8  872.04   234.7  870.14   244.6  868.69   264.4  866.67   274.3  866.14
   276.5  866.16   291.5  866.51   432.4  872.38     472  873.49   481.9  875.65
   491.7  880.05   511.5  890.81   531.3  900.03   560.9   913.2   600.5  929.09
   620.2  937.44     640   946.4   659.8   955.8   719.1  984.99   798.2  1020.3
#Mann= 3 , 0 , 0
       0      .1       0   276.5    .045       0   291.5      .1       0
Bank Sta=276.5,291.5
XS Rating Curve= 0 ,0
Exp/Cntr=0.3,0.1

Type RM Length L Ch R = 1 ,11468.5 ,341.1,350.3,359.5
XS GIS Cut Line= 3
     1931617.027      439897.257     1931716.817      440004.175
     1932200.113      440401.637
#Sta/Elev= 30
       0  991.82    48.8  964.38    58.5  957.72    68.2  948.51      78  937.26
   107.2  899.85     117   887.9   126.8  877.84   136.5  872.16   146.2  870.18
   166.1  868.14   219.8  861.18   225.7  860.71   234.8  860.79   285.3  863.54
     325  862.55     335  863.28   374.7  869.04   434.3  871.17   444.2  871.98
   454.2  873.76     484  881.05   493.9  885.44   513.8  895.69   523.7  900.27
   613.1  937.79   672.7  966.71   732.3  997.25   752.1 1006.34     772  1014.4
#Mann= 3 , 0 , 0
       0      .1       0   219.8    .045       0   234.8      .1       0
Bank Sta=219.8,234.8
XS Rating Curve= 0 ,0
Exp/Cntr=0.3,0.1

Type RM Length L Ch R = 1 ,11118.4 ,279.3,286.7,297.3
XS GIS Cut Line= 3
     1931260.442      439789.967     1931628.907      440486.492
     1931735.825      440674.192
#Sta/Elev= 30
       0 1133.99    29.9 1115.44    79.8 1081.86   159.6 1022.62   199.5  994.66
   229.4  975.61   289.3  943.54   309.2  929.61   349.1  899.88     369  887.23
     379  881.82     399   873.2     409     870   448.8  861.91   563.3  851.18
   578.3  850.75   628.4  856.78   758.1  860.26     768  861.09     778  863.94
     788  869.44   807.6  884.79   827.3  903.34   866.5  943.76   886.2  960.75
     896   967.3   915.6  978.72   935.3   988.1   984.4 1004.48    1004 1013.11
#Mann= 3 , 0 , 0
       0      .1       0   563.3    .045       0   578.3      .1       0
Bank Sta=563.3,578.3
XS Rating Curve= 0 ,0
Exp/Cntr=0.3,0.1

Type RM Length L Ch R = 1 ,10831.4 ,303.3,299.9,291.4
XS GIS Cut Line= 3
     1931179.785       439815.41     1931262.126      440364.591
     1931264.967        440909.2
#Sta/Elev= 30
       0 1113.11    69.4 1069.17   168.6 1002.98   208.2  978.14   247.9  955.87
   317.3  920.11   347.1  903.25   366.9  890.69   376.8  885.38   386.7  881.66
   426.4  871.02   456.2  859.79   466.1  858.04   495.8   854.9   547.8  848.16
   555.3  847.86   562.8  848.03   674.1  854.74     694  857.99   713.8  862.15
   723.7  865.44   733.6  870.24   802.9  911.85   822.7  923.06   842.5  932.79
   882.1  950.61   971.2  981.93  1020.7  998.44  1040.5 1004.53  1099.9 1020.07
#Mann= 3 , 0 , 0
       0      .1       0   547.8    .045       0   562.8      .1       0
Bank Sta=547.8,562.8
XS Rating Curve= 0 ,0
Exp/Cntr=0.3,0.1

Type RM Length L Ch R = 1 ,10531.4 ,305,304.2,305.9
XS GIS Cut Line= 3
     1930809.092      439895.556     1930972.821      440421.409
     1931177.901      440927.154
#Sta/Elev= 30
       0 1109.28      20 1104.69      30  1101.1    60.1 1086.88   190.3  994.33
   260.4  950.77   350.5  892.62   380.5  875.57   410.6  861.58   430.6  855.24
   450.6  852.29   500.7  851.14   543.3  843.57   550.8  842.54   558.3  842.62
   610.3  847.47   699.6  852.99   709.5  854.45   719.4  857.25     779  880.69
   818.7     899   848.4   917.5   888.1  948.71     908   962.4   937.7  980.23
   967.5  995.69   997.3 1009.06    1027 1020.58  1056.8 1030.41  1096.5 1041.26
#Mann= 3 , 0 , 0
       0      .1       0   543.3    .045       0   558.3      .1       0
Bank Sta=543.3,558.3
XS Rating Curve= 0 ,0
Exp/Cntr=0.3,0.1

Type RM Length L Ch R = 1 ,10226.9 ,296.8,300,302.3
XS GIS Cut Line= 3
     1930495.973      439961.584     1930680.136      440474.605
     1930851.203      440998.629
#Sta/Elev= 30
       0 1011.08    19.8 1003.85    59.5  992.21    89.2  982.06   128.8  970.86
   198.2  945.48   247.8  931.17   277.5  920.23   366.7  889.46   386.5  884.31
   416.2  878.29   426.2  875.71   505.4  850.88   537.6  839.48   545.1  837.81
   552.6  837.49   554.9  837.39   604.1  840.97   623.8  843.36   682.9  853.05
   722.3   860.6   732.1  863.14   751.8  870.54   771.5  879.39   810.8   898.6
   869.9  926.04   909.3  942.74   958.5  962.68  1047.1  995.16  1096.3 1013.97
#Mann= 3 , 0 , 0
       0      .1       0   537.6    .045       0   552.6      .1       0
Bank Sta=537.6,552.6
XS Rating Curve= 0 ,0
Exp/Cntr=0.3,0.1
